HEC-RAS study DRPLKCR.prj: DRPLKCR

--- DRPLKCR.g01 (geometry) --- (continued)

Type RM Length L Ch R = 1 ,24949   ,497.1,523.5,550.4
XS GIS Cut Line= 4
     2101191.306      182284.406     2101161.358      182819.562
     2101201.723      182837.791      2101162.66      183387.271
#Sta/Elev= 30
       0 2212.41    29.4 2206.66    68.6 2194.56   126.72184.376   186.3 2174.43
   238.6 2160.09   274.5 2152.84   454.3 2129.71   477.2 2124.76   487.72120.842
   513.1 2122.14   539.2 2119.46  547.522115.842   551.8 2115.06   561.3 2115.77
  564.822118.631  566.522119.431  604.14 2121.55   659.92119.163   698.3 2119.27
  722.592121.575  727.952121.736   734.4 2123.18   757.4 2134.09   803.2 2159.23
   829.5 2171.49   937.7 2227.47   983.6 2248.11  1052.4 2281.73  1131.2  2313.9
#Mann= 11 ,-1 , 0
       0     .12       0   126.7     .06       0   487.7    .016       0
  547.52    .045       0   561.3    .016       0  564.82     .12       0
  566.52     .06       0  604.14     .12       0   659.9     .04       0
  722.59     .06       0  727.95     .12       0
#XS Ineff= 2 , 0
                          603.26         2123.95
Permanent Ineff=
       F       F
Bank Sta=547.52,561.3
XS Rating Curve= 0 ,0
Exp/Cntr=0.3,0.1

Type RM Length L Ch R = 1 ,24425.5 ,553.9,543.4,525.7
XS GIS Cut Line= 3
     2100741.031      182309.294     2100690.236      182898.172
      2100641.93      183434.511
#Sta/Elev= 30
       0 2182.43    42.4 2173.94   195.9 2148.39   313.5 2134.82   339.6 2132.86
   378.8 2127.67   401.7 2126.52   421.3  2123.2   444.1 2120.93   450.6 2118.36
  456.012117.595  484.882117.462   542.1 2111.15   583.6 2110.17   591.1 2109.29
   597.6 2110.01   617.2 2108.42   623.7  2110.1   672.7 2143.49   698.8 2159.45
   731.4  2177.6   790.2 2209.32   806.5 2216.96   868.5 2249.16   917.4    2273
   959.9 2290.82  1008.8 2307.27  1034.9 2314.55  1087.2  2326.6  1129.6 2338.14
#Mann= 5 ,-1 , 0
       0     .12       0  456.01    .016       0  484.88     .12       0
   583.6    .045       0   597.6     .12       0
Bank Sta=583.6,597.6
XS Rating Curve= 0 ,0
Exp/Cntr=0.3,0.1

Type RM Length L Ch R = 1 ,23882   ,26.9,26.9,26.9
XS GIS Cut Line= 2
     2099957.102      182531.139     2100603.629      183434.177
#Sta/Elev= 30
       0 2201.09   10.822199.154    39.3 2194.55    75.4 2184.19   108.1 2171.45
   186.7 2136.96   209.7 2128.42   232.6 2122.43  283.442117.313   301.4 2114.79
   317.8 2115.68  336.852113.945   409.5 2108.56  415.382106.428   422.6  2103.8
   429.2 2106.41  466.172106.827   517.6 2107.16  539.782105.531   550.4 2102.33
   573.3 2110.44     593  2120.2   648.7 2153.84     819 2249.49   891.1 2286.25
   950.1 2314.09   999.2 2334.69  1041.8  2348.8  1077.9 2355.56  1110.6 2356.92
#Mann= 8 ,-1 , 0
       0     .06       0   10.82     .12       0  283.44    .016       0
  336.85     .12       0  415.38    .045       0   429.2     .12       0
  466.17     .04       0  539.78     .12       0
Bank Sta=415.38,429.2
XS Rating Curve= 0 ,0
Exp/Cntr=0.3,0.1

Type RM Length L Ch R = 1 ,23855.2 ,485.8,485.5,479.9
XS GIS Cut Line= 2
     2099934.966      182545.461     2100581.494        183448.5
#Sta/Elev= 30
       0 2200.53      112199.913    45.9 2194.21    88.5 2180.64   117.9 2167.61
   173.6 2139.59   193.3 2130.91     213 2124.51   232.6 2121.04  268.122119.106
   275.2 2118.67     285  2115.8  320.092115.122   406.2 2109.07  424.822104.864
   432.4  2103.4     439 2104.68   517.6  2105.9   537.3    2102   543.8 2102.67
     557 2107.83   579.9 2118.99   668.3 2172.72   769.9 2228.62   845.2 2268.76
   940.3 2315.96     996 2340.06  1051.6 2359.79  1074.6 2365.64  1110.6 2369.74
#Mann= 6 ,-1 , 0
       0     .06       0      11     .12       0  268.12    .016       0
  320.09     .12       0  424.82    .045       0     439     .12       0
Bank Sta=424.82,439
XS Rating Curve= 0 ,0
Exp/Cntr=0.3,0.1

Type RM Length L Ch R = 1 ,23369.7 ,341.5,350,361.3
XS GIS Cut Line= 3
     2099546.328      182808.171     2099906.273      183280.112
     2100311.175      183634.749
#Sta/Elev= 30
       0 2128.13    8.642127.793   115.6 2123.26  163.452121.792   190.2 2120.68
   232.8  2115.6   288.6 2113.02   311.5 2112.96   393.5 2107.83   413.2 2105.67
   495.2 2104.17   518.1 2100.83   570.6  2099.3   583.7 2096.91   593.5 2096.72
   596.8 2096.75   606.6 2097.05   613.1 2099.14   622.9  2107.2   632.7  2113.6
     724 2163.75   756.6 2179.49   792.5 2193.26   844.7  2208.4   870.8 2213.57
   939.3  2229.4  1007.8 2240.89  1040.4 2247.94  1095.9  2263.8  1131.8 2277.04
#Mann= 6 ,-1 , 0
       0    .016       0    8.64     .12       0   115.6    .016       0
  163.45     .12       0   583.7    .045       0   596.8     .12       0
Bank Sta=583.7,596.8
XS Rating Curve= 0 ,0
Exp/Cntr=0.3,0.1

Type RM Length L Ch R = 1 ,23019.7 ,394.2,394.4,395.8
XS GIS Cut Line= 3
     2099467.289      182860.355     2099644.146      183497.263
     2099824.215      183991.166
#Sta/Elev= 30
       0 2126.66   232.3 2115.23   245.4 2115.69  367.762107.599  375.752106.922
   428.7  2103.1   530.1 2098.05     589 2093.46   634.8  2094.4   651.2 2091.76
   654.5 2091.57  664.822091.911   670.8 2096.64   683.9    2114   696.9 2126.75
   703.4 2134.47     772 2191.54   801.4 2213.51   817.7 2226.98   863.4  2259.8
   896.1  2280.2   922.2  2294.3   948.4 2306.06   987.5 2319.94  1049.6 2337.47
  1098.6 2348.46  1121.4 2350.69  1134.5 2349.34  1163.8 2339.15  1186.7 2329.43
#Mann= 5 ,-1 , 0
       0     .12       0  367.76    .016       0  375.75     .12       0
   651.2    .045       0  664.82     .12       0
Bank Sta=651.2,664.82
XS Rating Curve= 0 ,0
Exp/Cntr=0.3,0.1

Type RM Length L Ch R = 1 ,22625.3 ,447.7,458.7,471.5
XS GIS Cut Line= 2
     2099110.877      182911.686     2099421.207      183988.075
#Sta/Elev= 30
       0  2126.8   70.672123.289   134.3 2120.21   157.2 2120.57  195.542118.926
  227.272117.316   242.4 2117.66   330.8 2113.09   389.8 2107.67   438.9 2101.38
   524.1 2099.14     547 2095.36   550.3 2093.86   556.8 2086.95  559.122085.677
   563.4 2084.87   573.2 2085.76   586.3 2088.92     606 2090.36   655.1 2087.86
   661.7 2089.74   694.4 2114.17   864.7 2226.88   989.2 2305.45  1018.7 2322.14
  1041.6 2333.14  1061.3  2339.8  1080.9 2341.42  1097.3 2335.72  1120.2 2323.66
#Mann= 6 ,-1 , 0
       0    .016       0   70.67     .12       0  195.54     .06       0
  227.27     .12       0  559.12    .045       0   573.2     .12       0
Bank Sta=559.12,573.2
XS Rating Curve= 0 ,0
Exp/Cntr=0.3,0.1

Type RM Length L Ch R = 1 ,22166.5 ,570.1,588.2,602.7
XS GIS Cut Line= 2
     2099093.516      182922.537     2098785.357      183927.311
#Sta/Elev= 30
       0 2127.11   16.752125.529   87.552120.485   163.7 2115.96   232.5 2114.27
   379.8 2115.49   497.6 2100.06   553.3 2095.84   605.7  2088.7   694.1 2084.96
   713.7 2082.89   733.4 2079.03   746.5 2079.71   756.3 2077.15   759.6 2076.98
  770.112077.186     776 2079.34   782.5  2084.5   802.1 2104.22   825.1 2124.68
   874.2 2162.67   887.3 2171.78   903.6 2185.29     920 2195.51   929.8 2199.29
   936.4 2199.57   952.8 2194.04   982.2 2178.92  1008.4 2162.07    1051 2127.43
#Mann= 5 ,-1 , 0
       0    .016       0   16.75     .06       0   87.55     .12       0
   756.3    .045       0  770.11     .12       0
Bank Sta=756.3,770.11
XS Rating Curve= 0 ,0
Exp/Cntr=0.3,0.1

Type RM Length L Ch R = 1 ,21578.3 ,862.6,847.9,832.3
XS GIS Cut Line= 3
     2099073.985      182911.686     2098624.766      183228.527
     2098509.749      183896.929
#Sta/Elev= 30
       0 2127.54    5.392127.614   29.292126.664   79.152124.281   137.4  2122.2
   170.2 2124.15   196.3 2118.18   235.6 2116.34   274.9  2103.7   323.9 2068.47
   359.9 2064.98   376.3 2065.01   405.7 2068.26   431.9 2067.17   448.3  2063.1
   497.4 2076.57   572.6 2086.57   598.9 2092.68     802 2172.98   877.4 2190.05
   890.5 2190.88   906.8 2187.53   962.6  2166.8    1051 2124.29  1064.1 2115.75
    1087 2093.31  1093.6    2091  1129.6 2112.12  1191.9 2127.69  1227.9 2142.91
#Mann= 6 ,-1 , 0
       0    .016       0    5.39     .06       0   29.29    .016       0
   79.15     .12       0   359.9    .045       0   376.3     .12       0
Bank Sta=359.9,376.3
XS Rating Curve= 0 ,0
Exp/Cntr=0.3,0.1

Type RM Length L Ch R = 1 ,20730.4 ,505.2,510.7,513.3
XS GIS Cut Line= 2
     2098353.499      182729.395     2097999.766      183855.697
#Sta/Elev= 30
       0 2141.52    91.8 2127.55   160.7 2120.28   190.2 2115.71   209.9 2115.39
   252.5  2111.4     305 2109.37   406.6 2101.12   478.8 2087.45  523.372080.639
   534.5 2074.98  556.952075.942   570.6 2075.12   600.1 2063.29   616.5 2053.83
   626.3 2054.37   636.2 2052.46   695.2 2048.96   718.1 2044.61   724.7 2044.26
   731.3 2044.51   737.8 2046.72   757.5 2059.98   813.3  2089.7   865.7  2123.3
   901.8 2148.97   934.6 2170.76  1029.7 2227.33  1085.4 2256.28  1180.5 2298.09
#Mann= 5 ,-1 , 0
       0     .12       0  523.37    .016       0  556.95     .12       0
   718.1    .045       0   731.3     .12       0
#XS Ineff= 2 , 0
          695.25 2052.63
Permanent Ineff=
       F       F
Bank Sta=718.1,731.3
XS Rating Curve= 0 ,0
Exp/Cntr=0.3,0.1

Type RM Length L Ch R = 1 ,20219.7 ,356.4,352.7,350.7
XS GIS Cut Line= 3
     2098043.254      182647.938     2097763.197      183115.903
     2097532.524      183621.706
#Sta/Elev= 30
       0 2129.06   117.6 2115.74     147 2111.25     209    2099   254.7 2087.19
   293.9 2074.85     307 2068.78   336.4 2049.08  345.762049.559   372.3 2048.25
   378.8 2045.21   393.42044.225  489.91 2043.27  517.412041.635     529 2040.14
   532.3 2039.14  537.11  2035.7   542.1 2034.45   551.9 2035.52   558.4 2036.85
   571.5 2044.07   587.9  2056.6   627.1 2081.06   669.6 2109.66   744.8 2147.99
   800.4 2173.71   826.6  2184.5   924.7 2218.61  1052.2  2280.1  1101.3 2300.98
#Mann= 7 ,-1 , 0
       0     .12       0  345.76    .016       0   393.4     .12       0
  489.91     .06       0  517.41     .12       0  537.11    .045       0
   551.9     .12       0
Bank Sta=537.11,551.9
XS Rating Curve= 0 ,0
Exp/Cntr=0.3,0.1

Type RM Length L Ch R = 1 ,19867   ,367.4,348.3,332.2
XS GIS Cut Line= 3
     2097639.523      182477.659     2097422.509      183052.745
     2097415.999       183593.11
#Sta/Elev= 30
       0 2209.47    52.3 2216.56    78.5 2218.59    94.8 2217.05   117.7 2209.67
   163.5 2186.33   238.7 2138.19   300.8 2095.69   349.8 2059.06   379.3 2039.79
   389.1 2035.77  397.052036.242  429.772035.415   447.9 2034.33   454.5 2030.45
   464.3 2030.12   477.4 2029.71   480.6 2030.13   516.6 2035.94   526.4 2039.55
   539.5  2047.4   585.2 2079.38   640.9 2114.08   716.2 2149.96   817.7 2191.51
   889.8 2216.08     952 2233.94  1030.6 2252.28  1089.6 2270.23  1155.1 2283.91
#Mann= 5 ,-1 , 0
       0     .12       0  397.05    .016       0  429.77     .12       0
   464.3    .045       0   480.6     .12       0
Bank Sta=464.3,480.6
XS Rating Curve= 0 ,0
Exp/Cntr=0.3,0.1

Type RM Length L Ch R = 1 ,19518.8 ,352.9,348.4,340.9
XS GIS Cut Line= 3
     2096875.429      182538.409     2097147.731      182992.248
     2097353.927      183599.017
#Sta/Elev= 30
       0 2165.68    16.3 2163.25    35.9    2165   101.3 2160.67   186.2 2147.67
     245 2134.14   287.5 2120.11   297.3 2114.17   310.4 2112.01   362.6 2084.76
   385.5 2070.54   414.9 2045.19     428 2035.75   437.8 2030.54   447.6 2028.07
  473.142026.227  511.252025.675   529.3 2022.36   539.1 2022.13  542.772022.424
   552.2 2027.25   588.1 2028.04   594.6 2029.64   604.5 2037.13   650.2 2063.12
   715.6 2096.32   810.4 2140.59  1058.9 2247.51  1104.7 2261.52  1170.1 2275.41
#Mann= 5 ,-1 , 0
       0     .12       0  473.14    .016       0  511.25     .12       0
   529.3    .045       0  542.77     .12       0
#XS Ineff= 2 , 0
          476.09 2031.38  567.35         2030.41
Permanent Ineff=
       F       F
Bank Sta=529.3,542.77
XS Rating Curve= 0 ,0
Exp/Cntr=0.3,0.1

Type RM Length L Ch R = 1 ,19170.4 ,168.8,194,216.6
XS GIS Cut Line= 3
     2096556.267      182814.702      2096921.32      183221.246
     2097268.285      183662.383
#Sta/Elev= 30
       0 2309.24    65.4 2257.64   117.8 2218.04     193 2165.75   199.6 2159.51
   212.7 2154.92   238.8 2136.12   294.5 2101.13   333.7 2074.38   359.9 2054.46
   389.3 2034.38   405.7 2025.62   418.8 2021.63     445 2021.18   467.9  2017.5
   488.82018.618  522.162018.974   543.1 2015.93   549.6 2015.74   556.2 2015.94
     566 2018.03   588.8 2030.71   650.8 2071.91   706.3 2103.72   781.3 2144.49
   859.6 2183.56   921.6 2208.51   960.8 2220.75  1039.1 2240.58  1107.6 2253.89
#Mann= 5 ,-1 , 0
       0     .12       0   488.8    .016       0  522.16     .12       0
   543.1    .045       0   556.2     .12       0
Bank Sta=543.1,556.2
XS Rating Curve= 0 ,0
Exp/Cntr=0.3,0.1

Type RM Length L Ch R = 1 ,18976.4 ,33.2,33.1,36.5
XS GIS Cut Line= 4
     2096307.192      183057.843     2096810.056      183338.052
     2096792.869      183394.302     2097247.209      183667.705
#Sta/Elev= 30
       0    2317   124.3 2235.25   215.9 2180.01   238.8 2165.22   245.3 2159.46
   258.4 2154.46   268.2  2146.9   327.1 2111.03   418.7 2059.64   474.3 2023.66
   490.6 2017.91  516.47 2015.45  550.282018.285   569.1 2017.86   575.7 2014.74
  587.762013.612   598.5 2012.22   608.3 2011.65  613.352012.274   621.4 2017.46
  638.86 2017.59   670.5  2017.6     677 2019.12   775.2 2084.58   834.2 2120.01
   902.9 2155.31   948.7 2175.95  1017.4 2202.16  1082.9 2223.16  1164.7  2245.7
#Mann= 7 ,-1 , 0
       0     .12       0  516.47     .06       0  550.28    .016       0
  587.76     .12       0   598.5    .045       0  613.35    .016       0
  638.86     .12       0
Bank Sta=598.5,613.35
XS Rating Curve= 0 ,0
Exp/Cntr=0.3,0.1

Type RM Length L Ch R = 1 ,18943.3 ,396,357.2,315.5
XS GIS Cut Line= 4
     2096298.063      183071.278     2096776.419      183338.052
     2096759.232      183394.302     2097234.478      183680.002
#Sta/Elev= 30
       0 2319.11     141 2225.95   193.5 2194.94   232.9 2169.77   242.7 2161.54
   255.8 2157.11   275.5 2142.76   324.7 2112.15   403.4 2068.51   465.7 2027.45
   485.4 2018.23   511.6 2013.87  527.032015.692  539.152015.722   547.7 2016.46
   554.2 2013.92   570.6 2013.35   580.4 2012.31   583.7 2013.06   609.8 2017.72
  646.762017.213     675 2017.67   681.6 2020.03   795.7 2095.83   834.9 2119.01
     887 2145.64   939.2 2169.31  1017.5 2198.03    1073 2215.43    1161    2240
#Mann= 6 ,-1 , 0
       0     .12       0  527.03     .06       0  539.15    .016       0
   570.6    .045       0   583.7    .016       0  646.76     .12       0
Bank Sta=570.6,583.7
XS Rating Curve= 0 ,0
Exp/Cntr=0.3,0.1

Type RM Length L Ch R = 1 ,18586.2 ,467.8,472.2,475
XS GIS Cut Line= 3
     2096076.461      183594.752     2096618.241      183672.383
      2097151.42      183789.178
#Sta/Elev= 30
       0 2357.63    72.1 2302.71   137.6 2254.78     272 2160.72     426 2058.01
   458.8 2037.58   488.3 2020.86   501.4 2016.96   514.5 2010.23   524.4 2008.94
   534.2 2004.24     544 2003.84   553.8 2003.61  558.352003.822   563.7 2005.88
   570.2 2010.33  595.032011.314   609.4 2012.36   625.8 2011.76  631.042013.551
   642.1 2021.83   697.7 2053.82   730.3 2069.68   772.8 2087.78   838.2 2110.12
   910.1 2132.24   978.7 2150.89  1034.3 2162.88  1057.2 2172.29  1093.1 2191.98
#Mann= 5 ,-1 , 0
       0     .12       0     544    .045       0  558.35     .12       0
  595.03    .016       0  631.04     .12       0
Bank Sta=544,558.35
XS Rating Curve= 0 ,0
Exp/Cntr=0.3,0.1

Type RM Length L Ch R = 1 ,18113.9 ,293.4,305.2,316.5
XS GIS Cut Line= 3
     2096006.834      183962.629     2096527.388      184134.278
     2097037.796      184326.382
#Sta/Elev= 30
       0 2278.92    81.6 2226.75   104.4 2217.27   150.1 2201.83   212.1 2168.01
     248 2145.46   306.7 2105.59     385 2058.92     447 2019.78   463.3 2007.18
   479.6 2000.75     509 1999.41     522 1996.28   538.3 1994.92   541.6 1994.62
   551.4 1994.89  573.911999.318   593.8 2002.09  605.472002.405   629.8 2002.51
   639.6 2006.06   659.2 2007.08   665.7 2010.02  674.932018.862   685.3 2025.66
   812.6  2098.3   848.6 2115.91   910.6 2150.11   972.7 2188.78  1093.5 2267.71
#Mann= 6 ,-1 , 0
       0     .12       0   538.3    .045       0   551.4     .12       0
  573.91     .06       0  605.47    .016       0  674.93     .12       0
Bank Sta=538.3,551.4
XS Rating Curve= 0 ,0
Exp/Cntr=0.3,0.1

Type RM Length L Ch R = 1 ,17808.7 ,392.3,394.8,396.5
XS GIS Cut Line= 3
     2095963.078      184049.555     2096396.146       184395.61
     2096751.716      184808.891
#Sta/Elev= 30
       0 2231.94      23 2221.98    65.6 2196.46   173.8 2118.81   203.4 2100.36
   232.9 2079.31   249.3 2070.52   305.1 2046.34   318.2 2037.84   337.9 2020.17
   347.7 2013.91   357.5 2012.35   370.7 2003.79   393.6 1998.08   461.11996.354
  509.25 1995.19   564.1 1990.57   573.9 1989.35  578.651990.486  579.341990.793
   593.5 1998.89   603.3  1999.8   613.1 2003.87   632.7  2004.2   644.12010.713
     711 2032.83   776.3 2048.52   874.3 2075.86     969 2111.11  1099.5  2164.5
#Mann= 7 ,-1 , 0
       0     .12       0   461.1    .016       0  509.25     .12       0
   564.1    .045       0  578.65     .12       0  579.34    .016       0
   644.1     .12       0
#XS Ineff= 2 , 0
          502.87  1998.3
Permanent Ineff=
       F       F
Bank Sta=564.1,578.65
XS Rating Curve= 0 ,0
Exp/Cntr=0.3,0.1

Type RM Length L Ch R = 1 ,17413.9 ,355.9,350,342.9
XS GIS Cut Line= 3
     2095800.892      184241.614     2096124.973      184681.383
     2096446.087      185122.912
#Sta/Elev= 30
       0 2165.81   173.4 2106.32   222.4 2082.98   235.5 2074.94   251.9 2071.43
   307.5 2045.99   330.4 2036.64   343.5 2033.34   431.8  1994.5   444.9 1990.96
  468.561989.787  486.841988.979   520.1 1987.88   536.5 1981.66   546.3 1980.96
   552.8 1981.64  554.541982.389   562.6 1985.36   585.5 1985.69  595.481990.473
   634.6 2014.63     664 2035.77   690.1 2051.74   732.6 2073.27   814.4 2106.15
   830.7 2109.98     932 2143.82  1007.2 2165.18    1053 2174.89  1092.2 2180.58
#Mann= 7 ,-1 , 0
       0     .12       0  468.56     .06       0  486.84     .12       0
   536.5    .045       0   552.8     .12       0  554.54    .016       0
  595.48     .12       0
Bank Sta=536.5,552.8
XS Rating Curve= 0 ,0
Exp/Cntr=0.3,0.1

Type RM Length L Ch R = 1 ,17063.9 ,362.1,350,340
XS GIS Cut Line= 3
     2095434.697      184580.102     2095865.522      184913.644
     2096307.943      185244.622
#Sta/Elev= 30
       0 2234.97   101.1 2196.23   117.4 2186.86   133.8 2181.04   172.9 2161.98
   182.7    2159     261  2117.9   342.6 2070.66   450.2 2024.77   473.1 2009.68
   495.9 1991.06     509 1982.24   535.1 1976.59   544.8 1976.24   551.4 1976.68
  567.121979.934   577.5 1981.42  606.521981.119   639.7  1980.1   659.3 1981.85
   662.6 1983.25   682.2  1999.5     705 2013.86   780.2 2052.09   835.8 2074.82
   901.2 2096.48   930.6 2101.76   963.3 2104.77  1028.7 2107.54  1097.4    2107
#Mann= 5 ,-1 , 0
       0     .12       0   535.1    .045       0   551.4     .12       0
  567.12    .016       0  606.52     .12       0
Bank Sta=535.1,551.4
XS Rating Curve= 0 ,0
Exp/Cntr=0.3,0.1

Type RM Length L Ch R = 1 ,16713.9 ,340.2,350,353.5
XS GIS Cut Line= 3
     2095186.036      185165.385     2095727.595      185229.638
     2096266.273      185338.859
#Sta/Elev= 30
       0 2203.63    75.1  2186.7   117.6 2174.44   199.2 2144.61   241.7 2127.13
   267.8 2113.46   284.1 2107.12   342.9 2075.64   411.5 2035.35   457.2 2005.65
   493.1 1980.68   509.4 1973.95   525.8 1972.93  533.87 1970.92   538.8 1970.22
   548.6 1970.81  560.991974.269  570.531974.433  602.331974.725  632.471973.936
     637 1974.63     650 1981.26   695.8 1991.78   725.3 1994.84   790.7 2010.57
   843.1 2018.31     866 2024.02   898.7 2035.63   973.9  2048.3    1095 2077.19
#Mann= 7 ,-1 , 0
       0     .12       0  533.87    .045       0   548.6     .12       0
  560.99     .06       0  570.53    .016       0  602.33     .06       0
  632.47     .12       0
Bank Sta=533.87,548.6
XS Rating Curve= 0 ,0
Exp/Cntr=0.3,0.1

Type RM Length L Ch R = 1 ,16363.9 ,519.2,519.3,522.2
XS GIS Cut Line= 3
     2095156.447      185279.904     2095648.835      185563.052
     2096154.589      185758.258
#Sta/Elev= 30
       0 2188.84    39.2  2179.1    75.1 2167.82   176.3 2135.27   202.4 2124.93
   225.2 2113.84   248.1 2098.96   352.6 2039.64   411.3 2003.03   434.2  1986.6
   463.5 1972.15   476.6 1969.26   515.8 1969.28   532.1 1967.58   551.7 1967.97
   560.5 1966.31   564.7 1966.06   575.5 1966.26  577.791966.459   587.6 1970.03
   610.4  1970.3  619.081975.472   643.1 1992.32   688.8 2015.16   721.5 2026.74
   783.5 2044.42   806.4 2047.83   848.8  2058.3  1061.1 2101.36  1110.1 2108.22
#Mann= 5 ,-1 , 0
       0     .12       0   560.5    .045       0   575.5     .12       0
  577.79    .016       0  619.08     .12       0
#XS Ineff= 2 , 0
                          598.14         1972.47
Permanent Ineff=
       F       F
Bank Sta=560.5,575.5
XS Rating Curve= 0 ,0
Exp/Cntr=0.3,0.1

Type RM Length L Ch R = 1 ,15844.7 ,376.8,401,424.5
XS GIS Cut Line= 3
     2095119.992      185420.367     2095265.391       185932.52
     2095896.902      186290.593
#Sta/Elev= 30
       0 2173.44    52.3 2164.04   140.4 2142.13     245 2122.21   316.8 2106.36
     392 2084.94   476.9 2047.67   538.9 2025.27   561.8 2015.18   617.4  1984.9
   646.8 1964.03   665.3 1957.53   669.7 1957.26  677.931957.587  679.151957.757
   689.4 1959.86  720.381959.965   741.7 1960.22  754.331962.555   777.6 1962.66
  785.091964.831   797.3  1969.3   901.9 2029.02   960.8 2056.75   996.8 2077.48
  1065.4 2106.09  1130.8 2124.16    1157 2129.18  1202.8 2133.87  1258.4 2133.53
#Mann= 7 ,-1 , 0
       0     .12       0   665.3    .045       0  677.93     .12       0
  679.15     .06       0  720.38     .08       0  754.33    .016       0
  785.09     .12       0
Bank Sta=665.3,677.93
XS Rating Curve= 0 ,0
Exp/Cntr=0.3,0.1

Type RM Length L Ch R = 1 ,15443.7 ,497.5,511.4,524.6
XS GIS Cut Line= 2
     2095100.461      185431.218     2095104.801      186776.704
#Sta/Elev= 30
       0 2174.11   160.4 2131.42   252.1  2124.1   301.2 2115.27   366.7  2092.2
   402.7 2076.09   435.4  2068.1   556.5 2028.96   684.2 1983.99   739.9 1974.87
   756.2  1967.7   772.6 1954.72   826.2 1950.64   834.8 1949.94  839.761950.551
   851.2  1953.9   872.91952.675   893.7 1955.76  915.491954.935  945.021955.324
 1004.231954.277 1082.111956.511 1162.561962.911  1181.8 1971.11 1210.671973.723
 1241.251981.333  1250.6 1984.77  1276.8 1985.13  1312.8  1999.5  1345.5 2006.81
#Mann= 11 ,-1 , 0
       0     .12       0   826.2    .045       0  839.76     .12       0
   872.9    .016       0  915.49     .12       0  945.02     .06       0
 1004.23     .12       0 1082.11     .06       0 1162.56    .016       0
 1210.67     .06       0 1241.25     .12       0
#XS Ineff= 2 , 0
                          896.17         1959.87
Permanent Ineff=
       F       F
Bank Sta=826.2,839.76
XS Rating Curve= 0 ,0
Exp/Cntr=0.3,0.1

Type RM Length L Ch R = 1 ,14932.3 ,326.5,318.3,309.8
XS GIS Cut Line= 2
       2095083.1      185444.239     2094421.207      186414.291
#Sta/Elev= 30
       0 2170.83    45.9 2155.74   124.6 2134.39     164 2127.07   229.6 2120.97
   255.9 2112.75   305.1 2090.18   341.2 2070.99   360.8 2064.65   419.9 2031.68
   446.1 2019.26     538 1971.42   551.1 1964.07   570.8  1950.4  586.081943.216
     597 1942.68   602.1  1943.1  629.981947.688  663.56 1946.09  689.571945.214
  804.081944.931   846.3 1944.06   973.71945.433   984.1 1943.02  1010.3 1948.86
  1039.9 1948.13  1066.1 1957.68  1082.5 1960.02  1125.2 1976.46  1174.4 1991.04
#Mann= 8 ,-1 , 0
       0     .12       0  586.08    .045       0   602.1     .12       0
  629.98    .016       0  663.56     .12       0  689.57    .016       0
  804.08     .06       0   973.7     .12       0
#XS Ineff= 2 , 0
                          627.59         1950.28
Permanent Ineff=
       F       F
Bank Sta=586.08,602.1
XS Rating Curve= 0 ,0
Exp/Cntr=0.3,0.1

Type RM Length L Ch R = 1 ,14613.9 ,345.7,350,347.8
XS GIS Cut Line= 3
     2094575.726      185295.593     2094451.872      185826.773
     2094328.768      186360.113
#Sta/Elev= 30
       0 2169.52    42.5 2154.39    71.8 2139.89   133.9 2103.88   192.7 2076.56
   254.8 2050.83   280.9  2032.8   336.4 2001.14     356 1988.22     418 1958.81
   437.6 1950.43   463.8 1943.08   493.2 1940.98   525.8  1941.3   537.9 1938.67
   545.4 1938.38     552 1938.61   565.1 1941.53   594.6 1939.91  617.281940.829
  648.291940.223   738.8 1941.55  838.151940.475  884.881942.245   899.4 1944.78
   909.2 1949.02   955.1 1981.28   997.7 2003.51  1053.5 2029.13  1092.8 2042.04
#Mann= 7 ,-1 , 0
       0     .12       0   537.9    .045       0     552     .12       0
  617.28    .016       0  648.29     .12       0  838.15     .06       0
  884.88     .12       0
#XS Ineff= 2 , 0
                          567.71         1944.41
Permanent Ineff=
       F       F
Bank Sta=537.9,552
XS Rating Curve= 0 ,0
Exp/Cntr=0.3,0.1

Type RM Length L Ch R = 1 ,14263.9 ,201.8,203.6,210.8
XS GIS Cut Line= 3
     2094332.604      185251.212     2094105.668      185793.821
     2094028.303      186326.796
#Sta/Elev= 30
       0  2107.8   111.1 2069.89   163.4 2046.69   205.8 2025.37   245.1 2000.48
   267.9 1983.06   300.6  1961.5     317 1953.22   333.3 1942.92   339.8 1941.56
   349.6 1937.06   359.4 1935.78  419.951936.561  502.081936.374   558.8 1936.46
   584.9 1933.01  600.081932.999   607.7 1934.39   624.1 1931.81   630.6 1933.29
   646.9 1942.38     660 1947.69   689.3 1954.84   780.7 1961.38   859.1 1974.73
   973.3 2019.86  1025.5 2044.96  1087.6 2071.89  1103.9 2076.62  1126.7 2085.67
#Mann= 5 ,-1 , 0
       0     .12       0  419.95     .06       0  502.08     .12       0
   584.9    .045       0  600.08     .12       0
Bank Sta=584.9,600.08
XS Rating Curve= 0 ,0
Exp/Cntr=0.3,0.1

Type RM Length L Ch R = 1 ,14060.3 ,543.9,530,512.1
XS GIS Cut Line= 2
     2094197.683      185179.482       2093687.7      186171.235
#Sta/Elev= 30
       0 2047.17    29.5 2040.52    52.5 2037.31    95.1 2027.61   200.1  1998.4
   278.8 1972.24   295.2 1963.74   321.4 1944.66     328 1941.74   354.2  1936.5
   416.41933.969   462.5  1932.1  502.451932.194   564.2 1931.94   583.8 1929.64
   590.4 1929.17   600.2 1929.57   610.1 1933.26     633 1935.89   665.8 1946.88
   701.9 1956.68   800.3    1976   888.9 2005.56   928.2 2019.79     984 2041.89
    1007 2048.24  1029.9 2049.67  1039.8 2047.84    1066 2039.34  1115.2 2011.54
#Mann= 5 ,-1 , 0
       0     .12       0   416.4     .06       0  502.45     .12       0
   583.8    .045       0   600.2     .12       0
Bank Sta=583.8,600.2
XS Rating Curve= 0 ,0
Exp/Cntr=0.3,0.1

Type RM Length L Ch R = 1 ,13530.3 ,363.2,371.3,378.4
XS GIS Cut Line= 2
     2093464.176      184945.107      2093679.02      186186.426
#Sta/Elev= 30
       0 2038.04    91.9 2023.14   213.2 1998.55   301.8  1979.4   311.7 1975.81
   337.9 1971.01  390.261958.289  395.451957.317     479 1943.54   495.4 1937.39
   518.3 1924.43   524.9 1922.14   534.8 1921.68   541.3 1922.07  578.451926.259
  612.921927.092   793.9 1927.91  878.661930.117   892.3 1932.19   915.3 1938.74
     958 1955.44  1007.2 1979.12  1053.1 2004.58  1095.7  2026.1  1131.8 2041.68
  1154.8 2048.71  1171.2  2049.9  1194.2 2042.86  1220.4 2028.46  1259.8 2002.99
#Mann= 8 ,-1 , 0
       0     .12       0  390.26     .06       0  395.45     .12       0
   524.9    .045       0   541.3     .12       0  578.45     .08       0
  612.92     .06       0  878.66     .12       0
#XS Ineff= 2 , 0
                           745.6         1930.33
Permanent Ineff=
       F       F
Bank Sta=524.9,541.3
XS Rating Curve= 0 ,0
Exp/Cntr=0.3,0.1

Type RM Length L Ch R = 1 ,13159   ,302.8,296.2,285.4
XS GIS Cut Line= 2
     2093288.395      184940.766     2093099.593      186023.666
#Sta/Elev= 30
       0  2029.5    49.1 2006.97   130.9 1976.15   166.8 1961.29   183.2 1956.32
   189.8 1953.06   199.6 1950.86   215.9 1949.15  238.351948.659   317.3 1951.25
   363.1 1949.63   392.6 1947.12  396.641946.019   402.4 1942.99     422 1927.22
   431.8  1922.5   438.4 1921.19   454.7 1920.49   477.6 1916.34   487.5 1916.07
   490.7 1916.35  503.561921.752   667.4 1921.99  792.171920.797  833.721919.872
     880  1919.6   974.9 1922.08 1055.821922.108  1079.6 1921.04  1099.2 1923.13
#Mann= 9 ,-1 , 0
       0     .12       0  238.35     .06       0  396.64     .12       0
   477.6    .045       0   490.7     .12       0  503.56     .06       0
  792.17    .016       0  833.72     .06       0 1055.82     .08       0
#XS Ineff= 2 , 0
                          511.46         1923.88
Permanent Ineff=
       F       F
Bank Sta=477.6,490.7
XS Rating Curve= 0 ,0
Exp/Cntr=0.3,0.1

Type RM Length L Ch R = 1 ,12862.8 ,342.5,350,357.8
XS GIS Cut Line= 3
     2092850.995      184932.264      2092931.07      185498.166
     2093089.528      186017.026
#Sta/Elev= 30
       0 1978.55      62 1974.68   69.181973.645  115.721970.918   192.7 1967.14
  220.971963.674   359.2 1951.34   385.4 1947.32   411.5 1941.94  460.731933.791
   473.6 1932.85   480.1 1931.48   489.9 1926.92     503 1922.79   512.8 1917.46
  519.941916.686   545.4 1916.91   558.5 1913.89     564 1913.64   571.5    1913
     579 1913.65   584.6  1916.8   587.9 1917.62  720.381918.122  773.791918.456
   839.5 1918.57   973.5 1920.98 1046.121921.013  1068.3    1921  1114.1 1923.35
#Mann= 11 ,-1 , 0
       0     .06       0   69.18    .016       0  115.72     .12       0
  220.97     .06       0  460.73     .12       0  519.94     .06       0
     564    .045       0     579     .06       0  720.38    .016       0
  773.79     .06       0 1046.12     .08       0
#XS Ineff= 2 , 0
                          613.25         1920.25
Permanent Ineff=
       F       F
Bank Sta=564,579
XS Rating Curve= 0 ,0
Exp/Cntr=0.3,0.1

Type RM Length L Ch R = 1 ,12512.8 ,360.5,370.2,382.5
XS GIS Cut Line= 3
     2092704.249      184920.714     2092597.352      185471.546
      2092567.42       186015.03
#Sta/Elev= 30
       0 1983.52      62 1982.32    94.6 1983.54   166.4 1974.77  192.751970.287
  216.411965.388  290.671949.639   316.4 1941.04  339.091938.406   401.3 1926.38
   456.7 1922.26   482.8 1923.86   502.4 1918.52   528.5 1914.36   551.3 1909.01
   564.4 1908.82   567.7 1908.88   580.8 1911.96  609.081911.519  653.351912.802
     830 1914.47   856.2 1915.37  862.231916.969   869.3 1919.97   892.3 1921.92
  904.341930.917   967.7 1973.77  1033.3 2015.52  1075.9 2039.05  1105.4 2050.64
#Mann= 11 ,-1 , 0
       0     .12       0  192.75     .06       0  216.41     .12       0
  290.67    .016       0  339.09     .12       0   551.3    .045       0
   567.7     .12       0  609.08    .016       0  653.35     .06       0
  862.23    .016       0  904.34     .12       0
#XS Ineff= 2 , 0
                          684.83         1964.05
Permanent Ineff=
       F       F
Bank Sta=551.3,567.7
XS Rating Curve= 0 ,0
Exp/Cntr=0.3,0.1

Type RM Length L Ch R = 1 ,12142.6 ,46.4,46.4,46.5
XS GIS Cut Line= 2
     2092581.295      184872.435     2092001.868      185701.863
#Sta/Elev= 30
       0 1998.74    3.431999.246    55.7 2004.49   140.8 1993.49   209.6 1966.52
  250.891953.894   271.8 1944.55  303.981940.273  320.81 1936.41  340.141930.627
  351.68 1928.32   386.4 1925.28     406 1919.46     442 1914.69   514.1 1910.66
  526.841905.504   533.7 1905.18   540.3 1905.54  552.771907.968  556.28 1908.67
  596.421907.788  645.081908.431  647.731908.471  731.69 1910.15   841.5 1916.78
  859.331929.415   867.7 1934.68   890.6 1941.84     907 1943.64  1011.8 1926.75
#Mann= 16 ,-1 , 0
       0     .12       0    3.43     .06       0  250.89    .016       0
  303.98     .06       0  320.81     .12       0  340.14     .06       0
  351.68    .016       0  526.84    .045       0   540.3    .016       0
  552.77     .06       0  556.28    .016       0  596.42     .06       0
  645.08     .12       0  647.73     .06       0  731.69    .016       0
  859.33     .12       0
Bank Sta=526.84,540.3
XS Rating Curve= 0 ,0
Exp/Cntr=0.3,0.1

Type RM Length L Ch R = 1 ,12096.2 ,427.1,425.3,422
XS GIS Cut Line= 2
     2092541.191      184849.779     2091961.764      185679.206
#Sta/Elev= 30
       0 1999.66    3.992000.202    55.7 2003.79   134.2 1992.59   170.3 1980.67
   225.9 1956.64   242.3 1952.58  251.081948.225   255.4 1945.66   307.8  1937.3
   317.6  1939.3   330.7 1938.67  363.261932.513   383.1 1931.12  412.811925.696
     442 1913.33   510.8 1908.22   523.9 1905.14   527.2 1905.03   540.3 1905.14
   576.3 1907.17  692.341908.181  744.781910.116   792.4 1911.57  812.591914.625
   841.5 1916.74   862.11927.972   884.1 1932.65   933.2 1920.72  1011.8 1922.96
#Mann= 11 ,-1 , 0
       0     .12       0    3.99     .06       0  251.08    .016       0
  363.26     .06       0  412.81     .12       0   523.9    .045       0
   540.3    .016       0  692.34     .06       0  744.78     .12       0
  812.59    .016       0   862.1     .12       0
Bank Sta=523.9,540.3
XS Rating Curve= 0 ,0
Exp/Cntr=0.3,0.1

Type RM Length L Ch R = 1 ,11670.9 ,371.6,370.4,368.8
XS GIS Cut Line= 3
     2092241.932      184563.194     2091978.335      185030.139
     2091714.932      185570.872
#Sta/Elev= 30
       0 2016.99    3.512016.369    55.6 2006.82  101.332015.714  148.292028.656
  186.562035.676  216.132041.182  230.722044.573   274.6 2053.77  296.262048.993
   382.5 1989.61   454.5 1943.49     503 1901.18     510 1899.88   516.6 1901.05
   532.9 1903.44   597.91903.117  623.141903.384   668.21903.285     837 1906.69
   856.6 1909.25  871.721917.092   902.3 1918.88   923.41935.683     935 1945.38
  953.231955.689   990.6 1972.09 1023.111978.866  1075.6 1981.26  1137.7 1992.83
#Mann= 17 ,-1 , 0
       0     .06       0    3.51     .12       0  101.33     .06       0
  148.29     .12       0  186.56     .06       0  216.13     .12       0
  230.72     .06       0  296.26     .12       0     503    .045       0
   516.6     .12       0   597.9     .06       0  623.14     .12       0
   668.2     .06       0  871.72    .016       0   923.4     .06       0
  953.23     .12       0 1023.11     .06       0
#XS Ineff= 2 , 0
                          676.23         1906.62
Permanent Ineff=
       F       F
Bank Sta=503,516.6
XS Rating Curve= 0 ,0
Exp/Cntr=0.3,0.1

Type RM Length L Ch R = 1 ,11300.6 ,543.4,538.4,530
XS GIS Cut Line= 2
     2091827.891      184500.228     2091330.929      185524.534
#Sta/Elev= 30
       0 2024.82    62.2 2016.06     121 2004.52   179.9 2005.49   196.3 2001.73
     229 1985.44   251.9 1969.11   307.5 1917.69   327.2 1902.37   340.2  1897.9
   366.4 1898.53   374.6  1896.7   382.8 1896.45  388.141896.726   402.4 1898.56
  467.411898.412   552.9 1899.44   654.3 1908.08  705.941909.006  754.211910.287
  804.431913.406     867 1917.98   896.4 1922.13  913.611927.414     952 1939.02
  1001.1 1946.93  1017.4 1947.01  1043.6 1943.27  1076.3 1943.07  1138.5 1951.26
#Mann= 8 ,-1 , 0
       0     .12       0   374.6    .045       0  388.14     .12       0
  467.41     .06       0  705.94     .12       0  754.21    .016       0
  804.43     .06       0  913.61     .12       0
Bank Sta=374.6,388.14
XS Rating Curve= 0 ,0
Exp/Cntr=0.3,0.1

Type RM Length L Ch R = 1 ,10762.2 ,345.3,356,367
XS GIS Cut Line= 3
     2091225.965      184335.653     2091140.824      184899.535
     2091059.902      185439.782
#Sta/Elev= 30
       0 2026.07    72.1 2008.95     154 1986.79   222.9 1974.23   258.9 1964.27
   311.4 1936.92   357.2  1909.5   376.9 1899.55   399.8 1893.87  426.891892.648
  544.751893.996     567 1892.04   576.8  1891.8   580.1 1892.03   645.5 1894.98
  662.621905.748   671.7  1907.6   691.3 1907.45  702.541914.887   717.5 1918.85
   782.9 1928.68   874.5 1930.88   900.6 1934.71   926.8 1940.46   943.2 1941.64
   975.9 1949.03  1002.1  1952.9  1044.6 1965.94  1067.5 1966.36  1116.6 1962.37
#Mann= 7 ,-1 , 0
       0     .12       0  426.89     .06       0  544.75     .12       0
     567    .045       0   580.1     .12       0  662.62    .016       0
  702.54     .12       0
Bank Sta=567,580.1
XS Rating Curve= 0 ,0
Exp/Cntr=0.3,0.1

Type RM Length L Ch R = 1 ,10406.2 ,343.7,349.8,349.6
XS GIS Cut Line= 3
      2091135.64      184299.403     2090838.685      184771.359
     2090489.206      185192.051
#Sta/Elev= 30
       0 1987.24    39.4 1970.02    75.4  1956.4   144.3 1937.51   249.3 1922.89
   331.3 1906.82   370.6 1892.66  427.861889.565  540.141889.454  552.141887.528
   557.6  1887.2   565.1 1887.53   580.5 1890.84  592.231897.611   600.2 1900.09
   619.8 1901.31  636.211913.965   688.6 1937.22   718.1 1944.47   734.4 1944.17
   757.4 1940.32   770.5 1935.74   790.1 1924.86   796.7 1922.88   819.6 1932.37
   858.9 1940.29   924.4 1946.11     967 1944.65  1025.9 1961.24  1104.5 1988.64
#Mann= 7 ,-1 , 0
       0     .12       0  427.86     .06       0  540.14     .12       0
  552.14    .045       0   565.1     .12       0  592.23    .016       0
  636.21     .12       0
Bank Sta=552.14,565.1
XS Rating Curve= 0 ,0
Exp/Cntr=0.3,0.1

Type RM Length L Ch R = 1 ,10056.4 ,354.7,351.1,355.3
XS GIS Cut Line= 3
     2090980.959      184177.646      2090575.63      184556.672
     2090227.024      184974.924
#Sta/Elev= 30
       0  1940.6    55.5 1945.18   104.5 1960.69   163.2 1983.89   195.9 1991.64
   212.2  1992.1   225.2 1989.85   248.1 1982.18   352.6 1931.24   401.5 1893.84
   411.3  1888.1  483.761888.198  488.981888.222   535.4 1887.22   551.7 1883.67
   558.2 1883.07   564.8 1883.68   581.2 1888.31  595.141895.512   617.2  1895.7
  631.271906.969   679.6 1931.58   732.1 1951.66   758.3 1956.43   791.1 1958.23
   866.5 1968.71   928.9    1981  1007.6 1990.92  1069.9  2004.4  1099.4 2008.46
#Mann= 7 ,-1 , 0
       0     .12       0  483.76     .06       0  488.98     .12       0
   551.7    .045       0   564.8     .12       0  595.14    .016       0
  631.27     .12       0
Bank Sta=551.7,564.8
XS Rating Curve= 0 ,0
Exp/Cntr=0.3,0.1

Type RM Length L Ch R = 1 ,9705.3  ,348.6,350,345.6
XS GIS Cut Line= 3
     2090719.912      183827.361     2090398.651      184264.288
     2089958.873      184623.063
#Sta/Elev= 30
       0 2114.78    62.1 2099.96   114.4 2081.76   228.7 2037.78   297.3 2020.57
   326.7 2010.38   375.7 1985.62   447.6 1942.06   467.2 1932.93   480.2 1919.82
   509.6 1898.83     526  1884.1   534.8  1880.4   542.3 1880.16   548.9 1880.38
     562 1884.81  617.851884.177   686.7 1884.69  703.361887.698   716.2 1894.25
   739.2 1895.22  751.961906.811  759.691910.786   794.9 1927.45     831 1941.43
   939.3 1960.07  987.671963.365    1018 1965.06 1059.051963.165  1109.9 1966.19
#Mann= 9 ,-1 , 0
       0     .12       0   534.8    .045       0   548.9     .12       0
  617.85     .06       0  703.36    .016       0  751.96     .08       0
  759.69     .12       0  987.67     .06       0 1059.05     .12       0
Bank Sta=534.8,548.9
XS Rating Curve= 0 ,0
Exp/Cntr=0.3,0.1

Type RM Length L Ch R = 1 ,9355.3  ,349.2,350,354.6
XS GIS Cut Line= 3
     2090508.559      183595.426     2090163.104      184013.566
     2089790.254      184440.049
#Sta/Elev= 30
       0 2032.17    39.2 2003.85    81.7 1980.16      98  1973.3   166.6 1950.57
   199.3 1941.49   258.1 1932.43   320.2 1925.16   359.4 1924.53   395.4 1921.72
   434.6  1915.4   493.4 1900.98   509.7 1893.43   535.8 1877.38   548.9 1877.28
   552.2 1877.45   565.3 1880.16  631.83 1880.03   702.8 1881.23   745.4 1886.46
  762.311890.766   771.6  1892.6   791.2 1892.45  799.411895.245     8161897.577
   837.1 1900.09   915.7 1903.76     955 1908.89  1017.2 1922.09  1108.9 1951.16
#Mann= 7 ,-1 , 0
       0     .12       0   535.8    .045       0   552.2     .12       0
  631.83     .06       0  762.31    .016       0  799.41     .08       0
     816     .12       0
Bank Sta=535.8,552.2
XS Rating Curve= 0 ,0
Exp/Cntr=0.3,0.1

Type RM Length L Ch R = 1 ,9005.3  ,519.8,525.2,525.6
XS GIS Cut Line= 3
     2090237.309      183421.522     2089862.269      183843.546
     2089428.093      184169.178
#Sta/Elev= 30
       0 1999.06    22.8 1990.42    71.8 2005.28  119.652011.307   153.4 2006.69
   241.5 1984.88   267.6 1987.11     297 1986.32  339.931981.234     359 1974.35
   385.1 1961.62   427.5  1934.3   509.1  1892.5     545 1876.22   561.3 1874.28
   567.9    1874   574.4 1874.21   584.2 1877.97  604.441877.229   639.8 1875.98
   750.9 1879.29  797.171884.858   809.8  1889.1   839.2  1889.5  845.251892.223
  991.981938.308  993.421938.591  1028.8 1940.59 1054.691939.408  1107.3 1937.12
#Mann= 11 ,-1 , 0
       0     .12       0  119.65     .06       0  339.93     .12       0
   561.3    .045       0   574.4     .12       0  604.44     .06       0
  797.17    .016       0  845.25     .06       0  991.98     .12       0
  993.42    .016       0 1054.69     .06       0
Bank Sta=561.3,574.4
XS Rating Curve= 0 ,0
Exp/Cntr=0.3,0.1

Type RM Length L Ch R = 1 ,8480.2  ,281.2,283,284.2
XS GIS Cut Line= 2
     2089944.211      183141.721     2089041.433      183788.423
#Sta/Elev= 30
       0 1913.32    26.2 1920.49   38.991922.404    72.1 1925.92      95 1925.48
   212.9 1905.77   252.2 1908.63   281.7 1917.33   330.9 1924.72   350.5 1925.31
  380.271921.441   412.8  1903.9   458.6 1872.34   491.4 1869.78   497.9 1869.17
  506.77 1869.82   514.3 1872.14  527.221871.613   573.3 1872.17  655.491877.483
   779.6  1881.9  845.29  1888.3   858.3 1891.73  887.011893.548   897.6 1900.66
  919.851908.644   989.3 1935.67  1058.1 1956.07 1097.491965.025  1110.5 1965.07
#Mann= 11 ,-1 , 0
       0     .12       0   38.99     .06       0  380.27     .12       0
   491.4    .045       0  506.77     .12       0  527.22    .016       0
  655.49     .06       0  845.29    .016       0  887.01     .08       0
  919.85     .12       0 1097.49     .06       0
Bank Sta=491.4,506.77
XS Rating Curve= 0 ,0
Exp/Cntr=0.3,0.1

Type RM Length L Ch R = 1 ,8197.2  ,30.2,30.3,30.2
XS GIS Cut Line= 3
     2089813.326      182933.113     2089383.639      183201.342
      2089028.17      183772.956
#Sta/Elev= 30
       0 1989.85    16.3  1990.4    42.5 1983.66    75.2 1967.57   130.7 1945.94
   160.1 1928.14   205.9 1911.52   241.8 1891.91     317 1876.41   336.6 1878.86
   370.11876.978   395.4 1879.38  421.161876.816  448.621873.332   467.3 1868.06
   477.1 1867.56  481.651868.038   493.5 1870.96  555.131871.063  592.42  1871.3
  627.211870.751   803.9 1876.05   882.3 1886.85   905.31895.087   928.1  1894.5
  940.251904.049  972.911914.043    1062  1942.3 1164.171964.783  1179.7 1965.26
#Mann= 13 ,-1 , 0
       0     .12       0   370.1    .016       0  421.16     .06       0
  448.62    .016       0   467.3    .045       0  481.65    .016       0
  555.13     .08       0  592.42     .12       0  627.21     .06       0
   905.3    .016       0  940.25     .08       0  972.91     .12       0
 1164.17     .06       0
Bank Sta=467.3,481.65
XS Rating Curve= 0 ,0
Exp/Cntr=0.3,0.1

Type RM Length L Ch R = 1 ,8166.9  ,567.7,561.6,556.9
XS GIS Cut Line= 3
     2089799.003      182907.071     2089369.316        183175.3
     2089013.847      183746.915
#Sta/Elev= 30
       0 2012.69    19.6 2012.42      36 2007.04   160.1 1947.04   189.5 1933.67
   209.2 1927.98   284.3 1890.61   300.6 1886.86   320.3 1878.27   339.9 1873.96
   359.5 1875.97  433.981872.658   454.2 1871.78  468.041868.039   480.2 1867.36
   483.7 1868.01   493.5 1870.93  544.881870.629  610.131870.628   807.2 1874.74
   849.6 1879.28   888.8 1886.28  912.251895.032   934.6 1894.23  945.781901.314
   950.9    1905  970.921911.315  1071.8 1941.29 1176.431964.002  1179.7 1964.25
#Mann= 10 ,-1 , 0
       0     .12       0  433.98    .016       0  468.04    .045       0
   483.7    .016       0  544.88     .08       0  610.13     .06       0
  912.25    .016       0  945.78     .08       0  970.92     .12       0
 1176.43     .06       0
Bank Sta=468.04,483.7
XS Rating Curve= 0 ,0
Exp/Cntr=0.3,0.1

Type RM Length L Ch R = 1 ,7605.3  ,348.2,350,347.6
XS GIS Cut Line= 3
     2089291.561      182507.775     2088944.149      182929.757
     2088530.224      183292.229
#Sta/Elev= 30
       0 2059.14    16.4 2054.61    49.1 2041.56   176.7 1982.82   232.4 1963.46
   258.6 1956.77   317.5 1947.42   346.9 1946.51   366.6 1948.69   382.9 1948.34
   402.6 1943.23   422.2 1934.54     468 1906.96   494.2 1893.82     527 1866.14
   533.5 1862.43   539.1 1861.47   546.6 1861.25   553.1 1861.47   569.5 1864.22
  616.751864.244     694 1864.84  767.611869.427  800.071872.071  801.561872.178
  887.031879.467  1034.6 1887.33 1052.681889.814  1090.2 1890.37  1096.8 1891.75
#Mann= 9 ,-1 , 0
       0     .12       0   539.1    .045       0   553.1     .12       0
  616.75     .06       0  767.61     .12       0  800.07     .06       0
  801.56     .12       0  887.03     .06       0 1052.68    .016       0
Bank Sta=539.1,553.1
XS Rating Curve= 0 ,0
Exp/Cntr=0.3,0.1

Type RM Length L Ch R = 1 ,7255.3  ,349.2,349.6,346.8
XS GIS Cut Line= 3
     2089078.742      182283.934     2088701.315      182678.489
     2088325.807      183074.857
#Sta/Elev= 30
       0 1969.36    16.4 1976.43    42.5 1982.99    65.4 1984.05    88.3 1981.42
     121 1971.98   209.2    1937   238.7 1928.56   264.8 1919.65   320.4 1898.14
     327 1898.72   353.1 1909.76   389.1 1918.81   418.5 1920.82   441.4 1918.39
   447.9 1916.35   457.7 1911.36   487.2  1892.6   516.6 1876.78   532.9 1860.02
   539.5 1857.85   542.7 1857.75   555.8 1857.87   575.4 1860.81  631.041862.392
   755.2 1864.04   846.8 1866.89   941.6 1871.68  1026.6 1874.03    1092 1878.93
#Mann= 4 ,-1 , 0
       0     .12       0   539.5    .045       0   555.8     .12       0
  631.04     .06       0
#XS Ineff= 2 , 0
                          682.55         1865.54
Permanent Ineff=
       F       F
Bank Sta=539.5,555.8
XS Rating Curve= 0 ,0
Exp/Cntr=0.3,0.1

Type RM Length L Ch R = 1 ,6905.7  ,351.3,350.4,352.3
XS GIS Cut Line= 3
     2088834.842      182060.927     2088444.799      182441.097
     2088115.583      182886.106
#Sta/Elev= 30
       0 1886.28    35.9  1885.8   69.18 1889.32    81.5 1892.18   107.6  1893.4
   159.8 1892.51   195.7 1893.72   215.3 1896.17     274  1893.8   335.9 1899.81
   391.4 1900.24   453.4 1895.83   469.6  1891.4  498.091878.495   505.5 1873.94
   508.8 1871.03   515.3 1862.95   521.8 1857.74   541.4 1855.33   544.7 1855.15
  555.731855.369   564.3 1857.42  569.621857.423   587.2 1857.15  641.441859.487
  679.061859.891   793.6 1860.34   865.7  1861.9   944.3 1867.93  1098.2 1872.89
#Mann= 8 ,-1 , 0
       0     .12       0   69.18     .06       0  498.09     .12       0
   541.4    .045       0  555.73     .12       0  569.62     .06       0
  641.44     .08       0  679.06     .06       0
#XS Ineff= 2 , 0
                          733.13         1862.26
Permanent Ineff=
       F       F
Bank Sta=541.4,555.73
XS Rating Curve= 0 ,0
Exp/Cntr=0.3,0.1

Type RM Length L Ch R = 1 ,6555.2  ,354.2,351.1,346.1
XS GIS Cut Line= 3
      2088491.58      181830.324     2088154.975      182261.016
     2087784.241      182666.223
#Sta/Elev= 30
       0 2087.57    39.3  2065.1    91.6  2041.8   117.8  2034.3   137.5 2030.78
   176.8  2029.9   189.8 2026.57   202.9 2027.03   229.1 2021.14     275 2005.11
   308.91988.726  329.151977.687   376.4 1955.51   392.8 1946.41   405.9  1936.3
   415.7    1933   477.9 1887.39   507.4 1857.95   520.4 1854.33  554.211853.041
   556.4 1852.87     563 1852.72  570.131852.933   582.6 1855.67  598.671856.525
  622.761856.876   654.71857.094  866.071859.157  987.211863.819  1095.8 1867.51
#Mann= 11 ,-1 , 0
       0     .12       0   308.9    .016       0  329.15     .12       0
  554.21     .08       0   556.4    .045       0  570.13     .12       0
  598.67     .06       0  622.76    .016       0   654.7     .06       0
  866.07    .016       0  987.21     .06       0
#XS Ineff= 2 , 0
                          737.67         1860.58
Permanent Ineff=
       F       F
Bank Sta=556.4,570.13
XS Rating Curve= 0 ,0
Exp/Cntr=0.3,0.1

Type RM Length L Ch R = 1 ,6204.2  ,358.8,350,341.4
XS GIS Cut Line= 3
     2088157.264      181611.154     2087862.046      182070.379
     2087582.449      182539.809
#Sta/Elev= 30
       0 2017.64    22.9 2018.24      36 2017.11    52.3 2014.07    98.1 2002.93
   183.1 1980.58   228.8 1965.48   274.6 1960.49   313.8 1959.23   343.2 1954.65
   362.9 1949.95     389  1938.4   421.7 1925.92  442.151912.801   460.9 1898.95
  482.52 1880.64   500.2 1866.25   506.7 1859.09   513.2 1854.75   519.8 1853.15
  543.891850.439   545.9 1850.32   555.8 1850.38   568.8  1850.4   578.6 1852.83
  586.281852.854   614.6 1852.57   644.1 1854.12   850.2  1855.8  1092.3 1864.62
#Mann= 6 ,-1 , 0
       0     .12       0  442.15    .016       0  482.52     .12       0
  543.89    .045       0   555.8     .12       0  586.28     .06       0
#XS Ineff= 2 , 0
                          650.51         1857.64
Permanent Ineff=
       F       F
Bank Sta=543.89,555.8
XS Rating Curve= 0 ,0
Exp/Cntr=0.3,0.1
